--- LFRFBUCRV.prj (project) ---

Proj Title=LFRFBUCRV
Current Plan=p01
Default Exp/Contr=0,0
English Units
Geom File=g01
Flow File=f01
Plan File=p01
BEGIN DESCRIPTION:
----------MODEL BY WOOD PLC 2022----------
AFH study
Randolph County, WV
HEC-RAS Version: RAS 6.2
Vertical Datum: NAVD88
Projection: NAD 1983 StatePlane West Virginia S FIPS 4702 (US Feet)
Terrain: 1-meter LIDAR (FEMA Region III 3DEP collected 2016-2018)
Land Use: 2019 NLCD
Hydrologic Method:
WV SIR2010-5033 regression equations
Additional Model Notes:
Added shared XS with SALTBLKRN to establish backwater tie-in
END DESCRIPTION:
DSS Export Rating Curves= 0
DSS Export Rating Curve Sorted= 0
DSS Export Volume Flow Curves= 0
DXF OffsetX= 0
DXF OffsetY= 0
DXF ScaleX= 0
DXF ScaleY= 0

--- LFRFBUCRV.p01 (plan) ---

Plan Title=Floodplain
Program Version=6.20
Short Identifier=Floodplain
Geom File=g01
Flow File=f01
Subcritical Flow
K Sum by GR= 0
Std Step Tol= 0.01
Critical Tol= 0.01
Num of Std Step Trials= 20
Max Error Tol= 0.3
Flow Tol Ratio= 0.001
Split Flow NTrial= 30
Split Flow Tol= 0.02
Split Flow Ratio= 0.02
Log Output Level= 0
Friction Slope Method= 1
Unsteady Friction Slope Method= 2
Unsteady Bridges Friction Slope Method= 1
Parabolic Critical Depth
Global Vel Dist= 0 , 0 , 0
Global Log Level= 0
CheckData=True
Encroach Param=-1 ,0,0, 0
Mapping Interval=1HOUR
Computation Time Step Use Courant=        0
Computation Time Step Use Time Series=    0
Computation Time Step Count To Double=0
Computation Time Step Max Doubling=0
Computation Time Step Max Halving=0
Computation Time Step Residence Courant=0
Run HTab= 0
Run UNet= 0
Run Sediment= 0
Run PostProcess= 0
Run WQNet= 0
Run RASMapper=-1
UNET Theta= 0
UNET Theta Warmup= 0
UNET ZTol= 0
UNET ZSATol= 0
UNET MxIter= 0
UNET Max Iter WO Improvement= 0
UNET MaxInSteps= 0
UNET DtIC= 0
UNET DtMin= 0
UNET MaxCRTS= 0
UNET WFStab= 0
UNET SFStab= 0
UNET WFX= 1
UNET SFX= 1
UNET Gravity=32.174
UNET 1D Methodology=Finite Difference
UNET DSS MLevel= 1
UNET Pardiso=0
UNET DZMax Abort= 0
UNET Use Existing IB Tables= 0
UNET Froude Reduction=False
UNET Froude Limit= 0
UNET Froude Power= 0
UNET D1 Cores= 0
UNET WindReference=Eulerian
UNET WindDragFormulation=Hsu (1988)
UNET D2 Coriolis=0
UNET D2 Cores= 0
UNET D2 Theta= 1
UNET D2 Theta Warmup= 1
UNET D2 Z Tol= 0.01
UNET D2 Volume Tol= 0.01
UNET D2 Max Iterations= 20
UNET D2 Equation= 0
UNET D2 RampUpFraction=0.1
UNET D2 TimeSlices= 1
UNET D2 Turbulence Formulation=Non-Conservative (original)
UNET D2 Eddy Viscosity=0.3
UNET D2 Transverse Eddy Viscosity=0.1
UNET D2 Smagorinsky Mixing=0
UNET D2 BCVolumeCheck=0
UNET D2 Cores=0
UNET D2 SolverType=PARDISO (Direct)
UNET D2 Minimum Iterations= 2147483647
UNET D2 Maximum Iterations= 2147483647
UNET D2 Restart Number= 10
UNET D2 Relaxation Coeff=1.3
UNET D2 SOR Precondition Iterations= 10
UNET D2 ILUT Maximum Fill= 8
UNET D2 ILUT Tolerance=1E-08
UNET D1D2 MaxIter= 0
UNET D1D2 ZTol=0.01
UNET D1D2 QTol=0.1
UNET D1D2 MinQTol=1
Write IC File= 0
Write IC File at Fixed DateTime=0
Write IC File at Sim End=0
Echo Input=False
Echo Parameters=False
Echo Output=False
Write Detailed= 0
HDF Write Warmup=0
HDF Write Time Slices=0
HDF Flush=0
HDF Compression= 1
HDF Chunk Size= 1
HDF Spatial Parts= 1
HDF Use Max Rows=0
HDF Fixed Rows= 1
Calibration Method= 0
Calibration Iterations= 20
Calibration Max Change=0.05
Calibration Tolerance=0.2
Calibration Maximum=1.5
Calibration Minimum=0.5
Calibration Optimization Method= 1
WQ AD Non Conservative
WQ ULTIMATE=-1
WQ Max Comp Step=1HOUR
WQ Output Interval=15MIN
WQ Output Selected Increments= 0
WQ Output face flow=0
WQ Output face velocity=0
WQ Output face area=0
WQ Output face dispersion=0
WQ Output cell volume=0
WQ Output cell surface area=0
WQ Output cell continuity=0
WQ Output cumulative cell continuity=0
WQ Output face conc=0
WQ Output face dconc_dx=0
WQ Output face courant=0
WQ Output face peclet=0
WQ Output face adv mass=0
WQ Output face disp mass=0
WQ Output cell mass=0
WQ Output cell source sink temp=0
WQ Output nsm pathways=0
WQ Output nsm derived pathways=0
WQ Create Restart=0
WQ Fixed Restart=0
WQ System Summary=0
WQ Write To DSS=0
Sorting and Armoring Iterations= 10
XS Update Threshold= 0.02
Bed Roughness Predictor= 0
Hydraulics Update Threshold= 0.02
Energy Slope Method= 1
Volume Change Method= 1
Sediment Retention Method= 0
Sediment TS Multiplier= 1
Warm Up Method= 0
XS Weighting Method= 0
Number of US Weighted Cross Sections= 1
Number of DS Weighted Cross Sections= 1
Upstream XS Weight=0
Main XS Weight=1
Downstream XS Weight=0
Number of DS XS's Weighted with US Boundary= 1
Upstream Boundary Weight= 1
Weight of XSs Associated with US Boundary= 0
Number of US XS's Weighted with DS Boundary= 1
Downstream Boundary Weight= 0.5
Weight of XSs Associated with DS Boundary= 0.5
Percentile Method= 0
Sediment Output Level= 3
Mass or Volume Output= 0
Output Increment Type= 1
Profile and TS Output Increment= 1
Transport Output Increment 1
XS Output Flag= 0
XS Output Increment= 10
Read HDF5 Sediment Hotstart= 0
Sediment Hotstart Type= 0
Write Gradation File= 0
Read Gradation Hotstart= 0
Write HDF5 File= 1
Write Binary Output= 1
Write DSS Sediment File= 0
DSS Sediment Output Type= 1
SV Curve= 0
Specific Gage Flag= 0
Subcell Erosion Methods= 0
Subcell Deposition Methods= 0
Advection Scheme= 1
Matrix Solver= 0
Implicit Weighting Factor= 1
Maximum Outer Loop Convergence Iterations= 5
Convergence Maximum Absolute= 0.001
Convergence RMSE= 0.0001
Grain Fractions Max Abs Error= 0.001
Max Subgrid Regions= 1
Max Subgrid Length Scale= 3.402823E+38
Initial Layer Thickness= 3.402823E+38
Min Layer Thickness= 3.402823E+38
Max Layer Thickness= 3.402823E+38
Number of Layers= 5

--- LFRFBUCRV.f01 (steady flow) ---

Flow Title=Flow
Program Version=6.20
Number of Profiles= 1
Profile Names=P100yr
River Rch & RM=LFRFBUCRV,Main,59067
     727
River Rch & RM=LFRFBUCRV,Main,51094
     820
River Rch & RM=LFRFBUCRV,Main,49850
    1100
River Rch & RM=LFRFBUCRV,Main,46470
    1380
River Rch & RM=LFRFBUCRV,Main,43332
    1580
River Rch & RM=LFRFBUCRV,Main,38450
    2210
River Rch & RM=LFRFBUCRV,Main,29488
    2720
River Rch & RM=LFRFBUCRV,Main,20950
    3030
Boundary for River Rch & Prof#=LFRFBUCRV,Main            , 1
Up Type= 0
Dn Type= 3
Dn Slope=0.011957
DSS Import GetInterval= 0
DSS Import GetPeak= 0
DSS Import FillOption= 0

--- LFRFBUCRV.g01 (geometry) ---

Geom Title=Geometry
Program Version=6.20

River Reach=LFRFBUCRV       ,Main
Reach XY= 30
2200278.73800004607211.3369999982198444.58400001609805.658000007
2199932.54100002611963.3510000112200351.02106965613834.559169009
2201699.03819487615538.8161471042201651.70000003617170.974000007
  2200099.254357620262.2484249032198074.05100003      620444.934
2196425.20900002 622055.880000012195204.19800001624909.024000004
2195342.95200004625282.3869999952196693.15900001625475.493000001
2197050.34200004627741.4382644742196810.52000003      628351.125
2197834.85900003629490.3560000212197813.08347383630071.997526169
2200466.15600003631604.0310000182199650.29800001633396.292999998
2200717.65499999634881.2720000152201081.61300002637129.733999997
2199371.51400004639016.9490000162198919.34900002638628.738000005
2197584.01000002638572.893000022      2196820.97637434.586999998
2196055.59346808637301.4281430392193894.99747384635667.410789937
2191572.79484296 635971.498157712191266.40100001636361.943210736
2189083.77499999635865.7080000192186646.64366651636335.791738245

Type RM Length L Ch R = 1 ,59067   ,389.7,389.7,389.7
XS GIS Cut Line= 4
2200170.50396211607183.0220105532200253.25238602607214.263584123
 2200634.6059526 607354.859670762200725.36783104607284.825358905
#Sta/Elev= 30
       0 2704.64     6.1 2701.97    14.6 2695.87    18.9 2694.51    27.4 2694.68
    61.6 2678.31    87.3  2664.4    95.8 2656.74  100.372654.187   117.1 2653.41
  122.372654.188   133.5 2658.04     164 2659.37   177.8 2656.28   210.9 2658.38
   248.7 2664.64   273.7 2665.91   343.1 2674.72   404.5 2678.76   424.1 2682.58
   436.9 2686.81   466.9 2686.05   479.5 2687.21   494.9 2692.25   497.6 2695.44
     507 2702.06   530.4 2715.33   548.5 2716.86   589.3  2734.4   609.5 2740.47
#Mann= 3 ,-1,0
       0      .1       0  100.37    .045       0  122.37      .1       0
Bank Sta=100.37,122.37
XS Rating Curve= 0 ,0
Exp/Cntr=0.3,0.1

Type RM Length L Ch R = 1 ,58677   ,283.2,283.2,283.2
XS GIS Cut Line= 4
2199994.93646883607373.6392003852200072.07743989607462.000676336
2200145.01072163607624.6979971332200233.37219758607762.149181944
#Sta/Elev= 30
       0 2708.81       8 2703.84    20.1 2697.95    28.9 2694.42    36.6 2692.98
    50.5 2685.55      79 2674.12      95 2669.02   100.3 2667.85   111.4 2667.01
   119.8 2664.72   128.9 2660.21     150 2645.51   155.8 2644.29   165.2 2644.15
  174.292638.453   177.8 2637.74  191.432638.452   210.6 2641.96   222.7 2640.94
   240.8 2641.91   287.4 2647.97   292.3 2650.07   316.2 2665.62     358 2679.38
   393.2 2694.01   410.3 2703.52   445.8 2728.25   451.6 2730.43     459 2731.67
#Mann= 3 ,-1,0
       0      .1       0  174.29    .045       0  191.43      .1       0
Bank Sta=174.29,191.43
XS Rating Curve= 0 ,0
Exp/Cntr(USF)=0,0
Exp/Cntr=0.3,0.1

Type RM Length L Ch R = 1 ,58394   ,309,309,309
XS GIS Cut Line= 4
2199748.07811646607546.9326028972199835.04427425 607658.35951178
2200019.42244666607725.8758839082200128.67010633607845.617397829
#Sta/Elev= 30
       0 2708.64    30.2  2695.4    53.6 2683.89    67.2 2679.39    78.6 2673.55
      90 2672.36    99.3 2667.34   129.7 2655.98   139.8 2650.32   155.3 2646.27
   172.5 2631.73  186.192627.958   193.7 2627.18  204.412627.958   219.3 2630.06
     232 2630.07   257.6 2635.44   287.9 2639.46   300.3 2642.23   322.2 2643.84
     330 2645.58   363.8 2661.77   380.4 2667.96   385.9  2671.4   396.3  2680.6
   401.7 2683.46   455.9 2705.37   488.4 2722.17   493.8 2724.05   499.8  2724.3
#Mann= 3 ,-1,0
       0      .1       0  186.19    .045       0  204.41      .1       0
Bank Sta=186.19,204.41
XS Rating Curve= 0 ,0
Exp/Cntr=0.3,0.1

Type RM Length L Ch R = 1 ,58085   ,172,172,172
XS GIS Cut Line= 4
2199583.67975769 607724.493388792199695.66093201607844.134912477
2199762.11099251 607965.520832942199896.59964051 608107.62317432
#Sta/Elev= 30
       0 2687.06      30 2674.95    47.6 2669.15    94.2 2662.21     116 2662.33
   139.5 2657.89   174.2 2643.68   187.9 2640.37   198.3 2632.49   210.7 2620.04
  214.212617.684     221 2616.79  231.962617.684   248.2 2621.32   265.4 2619.94
   274.1 2620.57   281.6 2622.54   291.7 2629.22   307.3 2632.13   328.9 2647.25
   343.2 2655.83   362.4 2659.72   367.9 2662.98   378.9 2671.92   389.9 2682.52
   402.5 2690.48   430.8 2701.84   450.5 2704.16   462.4  2712.2   497.9 2724.72
#Mann= 3 ,-1,0
       0      .1       0  214.21    .045       0  231.96      .1       0
Bank Sta=214.21,231.96
XS Rating Curve= 0 ,0
Exp/Cntr=0.3,0.1

Type RM Length L Ch R = 1 ,57913   ,123.7,123.7,123.7
XS GIS Cut Line= 3
2199475.94017111607907.3401086792199534.39993047607961.902550751
 2199828.2576542608159.106805668
#Sta/Elev= 30
       0 2664.21    12.8 2661.96    21.3 2657.42    44.1 2648.36    76.9 2630.05
    86.9 2626.74   100.9 2624.32   106.2 2621.84   115.8 2621.42   129.7 2613.51
   144.7 2613.53   188.1 2613.13   200.7 2611.44     222 2614.13   236.6 2625.71
   241.1 2628.27   256.6 2633.57   265.2 2638.65   273.9 2645.97   284.4  2647.4
   289.2 2649.37   298.9 2659.35   314.2 2672.92   322.7 2679.02   361.5 2694.18
   377.6 2701.77   380.5 2702.58   392.1 2702.13   404.9 2710.39   433.9 2720.03
#Mann= 3 ,-1,0
       0      .1       0   129.7    .045       0   144.7      .1       0
Bank Sta=129.7,144.7
XS Rating Curve= 0 ,0
Exp/Cntr(USF)=0,0
Exp/Cntr=0.3,0.1

Type RM Length L Ch R = 1 ,57789   ,303,303,303
XS GIS Cut Line= 3
2199373.60101095607971.1310853822199686.37258456608209.566814136
2199766.31868184608248.838581225
#Sta/Elev= 30
       0 2671.01       9 2665.88    23.3  2663.1    48.5 2646.59    73.7 2632.66
    94.6 2619.57   108.9 2613.22     139 2613.89   155.1 2618.27   179.3 2618.79
     186 2617.24   200.2 2609.03   208.8 2607.32   217.4 2607.49   239.6 2606.84
  249.922607.488   257.3 2612.57   265.9 2621.25   277.3 2631.25     295 2640.63
   322.9 2662.59   325.1 2663.61   335.2 2664.45   365.8 2678.55     380 2686.17
   395.3 2687.21   399.8 2688.37   409.3 2695.26   435.4 2705.89   482.4 2722.52
#Mann= 3 ,-1,0
       0      .1       0   217.4    .045       0  249.92      .1       0
Bank Sta=217.4,249.92
XS Rating Curve= 0 ,0
Exp/Cntr(USF)=0,0
Exp/Cntr=0.3,0.1

Type RM Length L Ch R = 1 ,57486   ,372.2,372.2,372.2
XS GIS Cut Line= 3
2199226.58993237608194.2503598582199467.35858264608437.073631466
  2199551.939349608476.753077395
#Sta/Elev= 30
       0 2656.19    13.6 2650.84    36.3  2644.2    45.6 2636.73    60.5 2634.41
    85.2 2619.79    94.3 2615.49   116.3 2610.43   127.6 2608.96   139.3 2601.56
   144.6 2599.83   155.9 2600.33  164.742596.967   178.6 2595.94     187 2596.93
   201.1 2599.72   212.4 2597.51   218.2 2597.28   223.8 2598.78   240.9 2600.96
   246.5 2603.44   268.9 2616.41   297.4 2634.49   325.6 2653.95   342.9 2654.88
   351.6 2661.84   395.9 2679.07   409.1 2686.08   420.8 2689.14   435.4 2695.59
#Mann= 3 ,-1,0
       0      .1       0  164.74    .045       0     187      .1       0
#XS Ineff= 2 , 0
                         200.595            2604
Permanent Ineff=
       F       F
Bank Sta=164.74,187
XS Rating Curve= 0 ,0
Exp/Cntr=0.3,0.1

Type RM Length L Ch R = 1 ,57114   ,392.2,392.2,392.2
XS GIS Cut Line= 3
2199069.40857475608515.3449541912199258.31875359608667.718735019
2199367.31699351608710.629122157
#Sta/Elev= 30
       0 2632.38    15.7 2625.89    31.7 2617.48    54.9 2601.62    60.3 2598.66
    70.4 2594.29    79.4  2589.2    85.8 2587.56   106.3 2586.95   111.4 2585.31
  116.632582.001     124 2581.21  134.492582.001   151.2 2583.11   162.6 2582.13
   173.9 2584.75   183.4 2585.07   193.7 2584.09   200.4 2585.52   205.2 2588.04
   210.9 2592.82   225.9 2603.78   238.7  2616.1   242.2 2618.05   269.9 2629.82
   283.4 2630.64   290.4  2632.1   303.9 2638.72   352.2  2656.1   359.8  2659.4
#Mann= 3 ,-1,0
       0      .1       0  116.63    .045       0  134.49      .1       0
Bank Sta=116.63,134.49
XS Rating Curve= 0 ,0
Exp/Cntr=0.3,0.1

Type RM Length L Ch R = 1 ,56722   ,348.5,348.5,348.5
XS GIS Cut Line= 2
2198878.58076587608866.5268560882199167.78608144 609027.09791068
#Sta/Elev= 30
       0 2620.24       9 2614.29    15.5 2610.58    47.3 2589.31    52.2 2585.32
    63.1 2575.47    70.8  2569.5   74.262567.865    79.6 2567.16    93.3 2567.32
    95.82567.863   106.1 2569.72   111.6 2571.79   120.8 2571.72   123.7 2572.36
   125.4 2572.96   129.9 2576.79   134.5 2579.15   152.8 2583.26   171.1 2586.01
   189.4 2587.12   198.6 2587.07   209.1  2588.4   217.9 2588.82     226 2590.16
   236.2 2593.03   248.9 2595.17   297.3 2607.35   305.9  2610.3   330.8 2620.58
#Mann= 3 ,-1,0
       0      .1       0   74.26    .045       0    95.8      .1       0
Bank Sta=74.26,95.8
XS Rating Curve= 0 ,0
Exp/Cntr=0.3,0.1

Type RM Length L Ch R = 1 ,56373   ,359,359,359
XS GIS Cut Line= 2
2198678.57910988609113.1060168532198934.40073043609358.805199186
#Sta/Elev= 30
       0 2591.58    12.5 2583.47    23.2  2577.9      38 2567.59    46.3 2562.84
    52.1 2560.66    57.8 2559.91    71.9 2561.73    77.6 2561.61    98.3  2559.7
  110.632557.245   115.6 2556.52   127.82557.245   134.1  2559.7   146.4 2559.68
   156.8  2563.5   167.6 2562.77   173.7 2561.14   184.9 2561.63   190.8 2560.46
   207.4 2560.62   213.4 2561.51   235.1 2568.15   254.2  2572.9   275.6 2583.39
   290.6 2584.49   296.2 2586.57   311.9 2594.21   320.9 2596.87   354.7 2609.35
#Mann= 3 ,-1,0
       0      .1       0  110.63    .045       0   127.8      .1       0
Bank Sta=110.63,127.8
XS Rating Curve= 0 ,0
Exp/Cntr(USF)=0,0
Exp/Cntr=0.3,0.1

Type RM Length L Ch R = 1 ,56014   ,86.9,86.9,86.9
XS GIS Cut Line= 3
2198508.32027495609279.5088344762198526.49749286609454.464556857
2198757.12094509609569.208244913
#Sta/Elev= 30
       0 2570.64     9.7 2566.46    34.2 2553.46    41.9 2551.18    94.2 2551.25
   130.4  2549.4   166.6 2549.36   182.2 2548.67   191.1 2545.92   194.1 2545.67
   204.6 2547.92     209 2548.09   231.4  2546.2  238.792542.576   240.3 2541.83
   244.8 2541.53  250.032542.576   253.7 2544.52   258.2 2545.53   267.1 2544.99
   302.9 2544.79   319.4  2545.9   325.2 2547.06   334.1 2553.55   347.5 2562.11
   352.2  2564.3   361.6 2567.43   374.4 2573.77   392.2 2580.58   433.5 2592.25
#Mann= 3 ,-1,0
       0      .1       0  238.79    .045       0  250.03      .1       0
#XS Ineff= 1 ,-1
 259.685433.4888    2550
Permanent Ineff=
       F
Bank Sta=238.79,250.03
XS Rating Curve= 0 ,0
Exp/Cntr(USF)=0,0
Exp/Cntr=0.3,0.1

Type RM Length L Ch R = 1 ,55927   ,58.6,58.6,58.6
XS GIS Cut Line= 6
2198480.35412404609287.4865256842198491.98773332609465.123790571
2198537.52693642609541.6957740432198585.60667781609598.062886377
2198604.01845525609694.5092956642198730.07726031609674.302643862
#Sta/Elev= 30
       0 2567.71    33.8    2553    41.8 2551.11    53.8 2551.25    77.9 2548.68
    97.9 2550.29     138 2547.17     184 2546.26   204.5 2544.88   215.3 2541.88
   233.2 2543.71   266.5 2541.46   277.1 2542.05   288.5  2538.9     298 2537.84
   308.3 2538.94   314.3 2540.56   333.9 2539.78   381.4 2541.68   410.4 2549.47
   439.8 2550.07   448.2 2553.63   464.3 2557.33   472.5 2562.88   496.7 2565.87
   504.8 2569.42   529.1  2576.2   537.2 2579.97   549.4 2581.59   567.5 2587.54
#Mann= 3 ,0,0
       0      .1       0   288.5    .045       0   308.3      .1       0
Bank Sta=288.5,308.3
XS Rating Curve= 0 ,0
Exp/Cntr=0.3,0.1

Type RM Length L Ch R = 1 ,55869   ,176.4,176.4,176.4
XS GIS Cut Line= 6
 2198455.8967676609287.3763313342198444.70373033609486.318466339
2198490.24293343609562.8904498112198538.32267482609619.257562145
2198556.73445226609715.7039714322198736.05543261609687.888437445
#Sta/Elev= 30
       0 2565.71    37.9  2550.8    41.9 2550.02    70.1 2551.25      98 2547.88
     138  2545.5     150 2543.55   262.2  2540.9   297.5 2539.17   319.7 2539.89
   334.5 2538.84   346.8 2539.68  357.82 2536.69   375.2  2536.7   393.8 2540.43
   406.1 2540.92   414.6  2539.3   430.4 2539.96   450.2 2538.33   461.1 2534.84
   492.9 2537.02   501.3 2543.71   509.1 2548.37   517.2 2550.68   545.5 2562.11
   561.7 2566.01   573.8 2567.11   585.4 2571.95   606.5 2577.14   642.5 2588.33
#Mann= 4 ,-1,0
       0     .08       0      80      .1       0  357.82    .045       0
   375.2      .1       0
Bank Sta=357.82,375.2
XS Rating Curve= 0 ,0
Exp/Cntr=0.3,0.1

Type RM Length L Ch R = 1 ,55692   ,144.5,144.5,144.5
XS GIS Cut Line= 2
2198184.03084997609801.6050267842198735.86358685609695.893248026
#Sta/Elev= 30
       0 2570.24    16.4  2566.5    44.9 2563.63    65.4 2558.14   122.3 2549.39
   133.8 2545.44   146.8 2536.14   154.3 2533.51   214.9 2533.66   236.4 2532.91
   248.6 2530.77   256.7 2529.87   271.7 2530.87   293.4 2531.33   309.7 2533.98
   321.9 2531.82   369.6 2535.24   387.1 2533.53   395.2 2535.84   411.5 2535.66
   415.6  2537.1   424.3 2544.16   444.1 2553.25   464.4  2560.8   488.9 2567.61
   501.1 2568.66   516.6  2574.4   529.6 2577.16   541.8 2582.01   561.9 2587.42
#Mann= 5 ,-1,0
       0      .1       0     100     .08       0     200      .1       0
   248.6    .045       0   271.7      .1       0
Bank Sta=248.6,271.7
XS Rating Curve= 0 ,0
Exp/Cntr(USF)=0,0
Exp/Cntr=0.3,0.1

Type RM Length L Ch R = 1 ,55548   ,397.1,397.1,397.1
XS GIS Cut Line= 4
2198258.06263147610113.3194466552198389.50388047609940.765138601
2198629.58581591609803.7296600362198768.47827125609746.596883544
#Sta/Elev= 30
       0 2590.79     5.2 2589.99    90.1 2561.59   109.1 2558.88   125.9 2553.57
     150 2548.35   176.2  2546.8     210 2541.59   224.6  2535.8   238.4 2526.16
   250.8 2524.77   279.9 2528.09   289.1 2526.98   316.7 2527.99   327.1  2526.1
   350.5 2526.12   362.8 2528.78   385.5 2529.98   412.1 2530.07   425.9 2528.55
   435.5 2530.36   450.3 2530.84   464.1  2528.2   473.7 2531.89   487.1 2532.32
   509.5 2546.01     531  2553.9   589.2 2572.15   608.6 2574.92   643.5 2584.74
#Mann= 4 ,-1,0
       0     .08       0     210      .1       0   327.1    .045       0
   350.5      .1       0
#XS Ineff= 2 , 0
        297.2142    2530
Permanent Ineff=
       F       F
Bank Sta=327.1,350.5
XS Rating Curve= 0 ,0
Exp/Cntr=0.3,0.1

Type RM Length L Ch R = 1 ,55151   ,388.6,388.6,388.6
XS GIS Cut Line= 2
2198540.61530163610304.0502036162198914.09943616609936.056436527
#Sta/Elev= 30
       0 2570.44       5 2568.91    16.2  2560.8    33.1 2557.99      44 2552.56
    69.6 2543.11   128.5 2524.31   182.7 2517.88   192.2 2514.62   201.5 2513.61
     211  2515.2   235.2 2515.04   250.6 2516.07   260.6 2514.55   267.6 2513.68
   285.8 2514.52   302.6 2518.46   328.9 2518.26   340.3 2516.53   353.2 2516.36
     370 2518.51   391.6 2516.49   408.7  2517.5     426 2516.75   434.5 2517.83
     443 2520.83   459.8 2530.88   487.9 2553.17   504.8 2562.33   524.3 2576.14
#Mann= 4 ,-1,0
       0     .08       0      50      .1       0   260.6    .045       0
   285.8      .1       0
Bank Sta=260.6,285.8
XS Rating Curve= 0 ,0
Exp/Cntr=0.3,0.1

Type RM Length L Ch R = 1 ,54762   ,364.2,364.2,364.2
XS GIS Cut Line= 2
2198675.62675498610539.659586707 2199072.5521152610177.798304245
#Sta/Elev= 30
       0 2570.51    15.6 2563.68    49.5 2553.08    60.3  2551.1    70.1 2545.01
    84.3 2543.29    98.4 2534.65   122.4 2523.19   134.3 2519.92   149.4 2511.04
  161.852505.805   180.5 2504.93  189.522505.806   195.6 2507.39   211.5 2507.09
   217.4 2508.75   238.9 2508.07   312.4 2511.94   324.3 2510.21   347.6 2510.49
   364.6 2508.62   381.6 2510.43   406.7 2508.92   435.4 2510.98   446.7  2513.8
   454.9 2517.78   478.7 2537.68   487.9 2543.63     509 2550.14   537.1 2560.93
#Mann= 3 ,-1,0
       0      .1       0  161.85    .045       0  189.52      .1       0
Bank Sta=161.85,189.52
XS Rating Curve= 0 ,0
Exp/Cntr(USF)=0,0
Exp/Cntr=0.3,0.1

Type RM Length L Ch R = 1 ,54398   ,391.9,391.9,391.9
XS GIS Cut Line= 2
2198876.05427233 610834.58010669     2199284.446610463.891243402
#Sta/Elev= 30
       0 2591.74      14  2585.5    32.2 2572.81    48.8 2569.49    75.8 2557.36
    86.6 2554.29   108.2 2545.28   117.2 2538.72   142.7 2524.87     154 2517.39
   165.3 2507.78   178.4 2500.29     188 2499.74   219.1 2501.83   253.1  2499.6
  260.822496.561   272.9  2495.9  289.932496.561   298.4 2499.64   321.1 2498.86
   335.1 2497.21   349.4 2498.15   363.5 2497.32   372.9 2500.68   426.9  2508.3
     474 2517.78   518.8 2528.09   531.8  2532.5   540.4 2536.91   551.5  2538.3
#Mann= 5 ,-1,0
       0      .1       0     130     .05       0     140      .1       0
  260.82    .045       0  289.93      .1       0
#XS Ineff= 2 , 0
                        304.4914            2501
Permanent Ineff=
       F       F
Bank Sta=260.82,289.93
XS Rating Curve= 0 ,0
Exp/Cntr=0.3,0.1

Type RM Length L Ch R = 1 ,54006   ,394.8,394.8,394.8
XS GIS Cut Line= 2
2199100.88490344611062.4107280292199594.10793273610747.591572513
#Sta/Elev= 30
       0 2569.23    29.3 2556.49    46.9 2551.26    76.6 2536.93    93.1 2531.35
   101.8 2525.65   117.8 2522.87   133.6 2513.79   148.1 2502.69   165.2 2491.59
   173.3 2488.07   185.8 2486.61   203.2 2488.57     235 2488.57   240.2 2486.79
   255.3  2485.7  265.612486.798   287.1 2489.07     322 2487.94   355.1 2489.97
   368.2 2488.79   429.1 2490.74     450 2500.13   469.6 2513.81   485.5 2521.84
   530.6  2542.7   540.1 2545.32   549.6 2550.36   559.1 2552.22   585.1 2564.23
#Mann= 4 ,-1,0
       0     .05       0      50      .1       0   240.2    .045       0
  265.61      .1       0
Bank Sta=240.2,265.61
XS Rating Curve= 0 ,0
Exp/Cntr=0.3,0.1

Type RM Length L Ch R = 1 ,53611   ,346.4,346.4,346.4
XS GIS Cut Line= 3
2199245.22198011611349.5380097652199334.83141683 611343.32824892
2199751.39266059611072.633568628
#Sta/Elev= 30
       0 2563.07      31 2546.06    59.1  2533.3    75.1 2528.01    83.2 2522.04
     101 2519.18   105.7 2517.05   135.7 2495.01   153.1 2486.18     163 2479.61
  181.752476.916   196.4 2476.06  206.09 2476.91   229.8 2480.58   253.6 2479.02
   267.9 2479.91   310.9 2476.56   373.2 2480.01     392 2478.32   444.4 2479.88
   463.5 2478.76   468.3 2481.14   477.8 2489.49   488.5 2493.17   497.5 2501.85
   508.7 2507.06     529 2512.88   563.7 2531.16   572.3 2533.42   586.6 2540.18
#Mann= 5 ,-1,0
       0      .1       0      20     .05       0  119.82      .1       0
  181.75    .045       0  206.09      .1       0
Bank Sta=181.75,206.09
XS Rating Curve= 0 ,0
Exp/Cntr=0.3,0.1

Type RM Length L Ch R = 1 ,53265   ,312.8,312.8,312.8
XS GIS Cut Line= 3
2199434.65183339611630.0682511932199575.52527219611580.080901942
2199895.89873785611276.748578073
#Sta/Elev= 30
       0 2517.61    22.8 2509.84    82.3 2493.82   117.8 2485.85   124.1  2481.7
   133.2 2471.23   137.4 2468.68   153.7 2469.72   180.3 2468.06   211.4 2469.18
  218.972467.482     234  2466.6  246.872467.483     255 2469.56   279.3 2468.06
   290.6 2469.72   304.6  2469.4   315.6 2471.35   345.7 2471.79   365.2 2473.68
   381.7 2471.47   409.5  2471.8   421.3 2469.52   437.8 2470.17   467.9 2480.35
   497.4 2494.72   530.5 2503.38   548.1 2513.51   556.6 2514.52   590.7 2534.17
#Mann= 3 ,-1,0
       0      .1       0  218.97    .045       0  246.87      .1       0
Bank Sta=218.97,246.87
XS Rating Curve= 0 ,0
Exp/Cntr(USF)=0,0
Exp/Cntr=0.3,0.1

Type RM Length L Ch R = 1 ,52952   ,278.6,278.6,278.6
XS GIS Cut Line= 4
2199519.83286417611872.8807925392199651.64237219611811.840430291
2200026.01573581611717.0509686552200120.51455373611588.188199994
#Sta/Elev= 30
       0 2523.94     8.8    2520      18 2518.78    56.4 2502.19    79.7 2495.04
    90.4 2489.25   105.5 2486.45   123.6 2475.81     137 2464.54   145.8    2461
   191.2 2459.32   233.5 2462.68   252.8 2459.22   263.1  2459.2   273.7 2462.07
   286.2 2459.44   302.6 2459.66   315.8 2462.96   351.7 2461.75   376.9 2458.21
   397.5    2461   414.6 2458.66   460.7 2460.52     480 2458.06   504.8  2460.1
   529.5 2469.53   575.9 2477.48   658.8 2506.12   670.3 2507.51   691.2 2516.53
#Mann= 3 ,-1,0
       0      .1       0   252.8    .045       0   263.1      .1       0
#XS Ineff= 2 , 0
                        455.4829            2464
Permanent Ineff=
       F       F
Bank Sta=252.8,263.1
XS Rating Curve= 0 ,0
Exp/Cntr=0.3,0.1

Type RM Length L Ch R = 1 ,52673   ,318.5,318.5,318.5
XS GIS Cut Line= 4
2199654.99908208612043.7452358262199751.61707069611994.748685507
2200316.73747909611978.1736164222200408.49690298612008.220585077
#Sta/Elev= 30
       0 2501.35    38.5 2485.84    49.9 2479.53    59.6 2478.15      82 2469.98
   104.5 2455.53   132.9  2453.4   172.9 2454.25   180.9 2452.83   220.9 2455.99
   236.9 2452.84     261 2454.34  282.232451.983   296.9 2451.99     305  2453.5
     365 2453.15     377 2449.21     401 2451.99     413 2456.23     445 2458.34
   513.1 2461.65   525.1  2457.5   552.5 2458.61   569.1 2466.46   605.1 2471.62
   641.1 2480.86   677.3  2493.2     701 2494.25     720  2504.8   770.2 2519.71
#Mann= 4 ,-1,0
       0      .1       0  282.23    .045       0   296.9      .1       0
  703.69     .06       0
#XS Ineff= 2 , 0
                        340.5182            2454
Permanent Ineff=
       F       F
Bank Sta=282.23,296.9
XS Rating Curve= 0 ,0
Exp/Cntr=0.3,0.1

Type RM Length L Ch R = 1 ,52355   ,275.4,275.4,275.4
XS GIS Cut Line= 4
2199774.33859308612319.6664556442199935.66140203612294.672781018
2200140.15510351612098.1316123692200373.05070798612089.043003414
#Sta/Elev= 30
       0 2477.09    10.8 2472.45    31.8 2466.46    45.8 2461.11    74.7 2454.59
   155.7 2446.19  165.15 2443.77     176 2442.87   187.22443.771   197.2 2446.58
   258.3 2444.43     286 2448.59   317.4 2445.83   335.9 2448.53   350.1 2444.44
   374.8 2448.58   391.4 2447.85   446.9 2453.06   458.9 2452.32   466.9 2449.55
   501.8  2453.8     527 2450.79     531 2451.38     543 2457.26     551 2462.54
     563 2473.04     587 2474.82     595 2483.72     599 2486.77     680 2515.13
#Mann= 4 ,-1,0
       0      .1       0  165.15    .045       0   187.2      .1       0
  556.88     .06       0
#XS Ineff= 1 ,-1
 287.057679.9506    2454
Permanent Ineff=
       F
Bank Sta=165.15,187.2
XS Rating Curve= 0 ,0
Exp/Cntr(USF)=0,0
Exp/Cntr=0.3,0.1

Type RM Length L Ch R = 1 ,52079   ,335.6,335.6,335.6
XS GIS Cut Line= 2
2199818.18156153612557.1119440592200346.05477306612510.651877017
#Sta/Elev= 30
       0 2467.04    30.1 2458.39    94.4  2449.8   118.4  2445.5   150.6 2443.49
   175.2 2438.71   202.8 2437.94  206.17 2437.14   218.8 2436.11  224.08 2437.14
   226.9 2438.79   230.9 2439.67   238.9 2436.84     251 2435.22   283.1 2435.94
   299.1  2434.5   311.2 2437.68   355.4 2435.08   367.4 2436.74   383.5 2436.08
   391.5 2437.73   435.7 2466.97   447.7 2473.54   455.7 2481.25   463.8 2486.55
   479.8  2491.9   495.9 2499.57   507.9 2500.98     516 2505.93   529.9 2512.18
#Mann= 5 ,-1,0
       0      .1       0  206.17    .045       0  224.08      .1       0
     330     .06       0     430      .1       0
#XS Ineff= 2 , 0
                        248.5047            2440
Permanent Ineff=
       F       F
Bank Sta=206.17,224.08
XS Rating Curve= 0 ,0
Exp/Cntr=0.3,0.1

Type RM Length L Ch R = 1 ,51744   ,298.6,298.6,298.6
XS GIS Cut Line= 2
2199858.40822591612861.5747645772200359.41779455  612821.8121004
#Sta/Elev= 30
       0  2464.1      62  2444.5      86 2441.52    94.1 2438.34  108.24 2429.94
   114.1 2428.57   126.2 2428.78   130.2 2429.93   150.2    2432   206.4 2431.69
   222.5 2428.66   266.6 2430.78   278.6 2430.45   286.7 2428.91   326.8 2428.05
   338.8 2426.43   346.9  2427.2   350.9 2429.28   362.9 2438.13   370.9 2446.46
     383 2455.57     387 2457.72     395 2460.14     403  2463.9   414.7 2466.25
   431.1 2474.22   451.2 2480.38   479.3 2494.98   495.3 2497.85   502.6 2502.31
#Mann= 5 ,-1,0
       0      .1       0  108.24    .045       0   130.2      .1       0
     200     .06       0     290      .1       0
#XS Ineff= 1 ,-1
  201.84 502.585    2440
Permanent Ineff=
       F
Bank Sta=108.24,130.2
XS Rating Curve= 0 ,0
Exp/Cntr(USF)=0,0
Exp/Cntr=0.3,0.1

Type RM Length L Ch R = 1 ,51445   ,351,351,351
XS GIS Cut Line= 3
2199865.46600644613123.5749834752199993.94113929613129.952055108
2200349.69003929613040.492871524
#Sta/Elev= 30
       0 2471.14    18.7 2464.53    30.7 2462.75    46.8 2455.85    62.8 2454.94
   106.8 2443.81   118.9 2437.29   135.1 2436.52   143.3 2431.21   159.8  2424.9
   192.8 2421.08   206.9 2421.57   217.6 2420.49  226.23 2421.56   242.3 2423.75
   250.5 2427.43  262.14 2421.66   262.9 2423.07   279.4 2422.25   289.3 2424.78
   324.8 2421.98     366 2423.72   378.3 2427.97   389.6 2438.18   400.6 2446.48
   427.9 2459.69   436.2 2460.79   444.4 2466.01   480.5 2478.02   495.5 2484.91
#Mann= 5 ,-1,0
       0      .1       0   206.9    .045       0  226.23      .1       0
   289.3     .06       0   389.6      .1       0
#XS Ineff= 2 , 0
                           250.5            2430
Permanent Ineff=
       F       F
Bank Sta=206.9,226.23
XS Rating Curve= 0 ,0
Exp/Cntr=0.3,0.1

Type RM Length L Ch R = 1 ,51094   ,313.1,313.1,313.1
XS GIS Cut Line= 3
2199944.99535949613596.4063880642200106.65591013613526.978786295
2200403.50948499613208.966582641
#Sta/Elev= 30
       0 2464.68    12.2  2461.8    38.6 2459.52    77.5 2449.44   125.4 2439.29
   142.8 2433.64   164.5  2421.8   175.9 2417.36   216.7 2417.97   230.9 2414.44
   240.5 2416.06   271.7 2416.92     283 2414.55   298.8 2413.77  311.642414.552
   320.7 2415.98   371.6 2417.85   395.1  2414.4   424.4 2418.27   479.4 2416.96
   490.3 2417.87   498.1 2420.85   512.2 2431.03   518.2 2433.29   529.2 2442.75
   540.5 2448.92   572.4 2460.94   583.3 2461.46   591.5 2463.42     611 2463.63
#Mann= 5 ,-1,0
       0      .1       0     283    .045       0  311.64      .1       0
  385.94     .06       0  525.94      .1       0
#XS Ineff= 2 , 0
                        357.6812            2426
Permanent Ineff=
       F       F
Bank Sta=283,311.64
XS Rating Curve= 0 ,0
Exp/Cntr=0.3,0.1

Type RM Length L Ch R = 1 ,50781   ,282.4,282.4,282.4
XS GIS Cut Line= 4
2200080.00721103613799.0760296972200276.36604648613712.117116857
2200540.04791122613637.7812720112200669.08371737 613504.53777653
#Sta/Elev= 30
       0 2459.36    22.1 2453.13    61.4 2444.51    71.3 2441.08    87.7 2439.59
   118.3 2428.06   144.1 2421.59   162.7 2415.27   188.3    2411     197 2410.76
   210.2 2414.03   218.7 2414.49   233.2 2407.83   239.5 2407.62   247.8  2409.5
   279.7 2407.15   285.2 2406.41  297.08 2407.15   310.1 2408.76   355.9 2408.15
   393.3 2410.54   430.7 2409.32   443.1 2407.69   455.6  2408.5   484.7 2406.17
   492.1  2407.1   517.6 2416.66   552.1 2426.59   576.9 2429.32   674.2 2465.53
#Mann= 6 ,-1,0
       0     .08       0      80      .1       0   279.7    .045       0
  297.08      .1       0  394.75     .06       0  548.71      .1       0
#XS Ineff= 1 ,-1
   424.2 674.196    2412
Permanent Ineff=
       F
Bank Sta=279.7,297.08
XS Rating Curve= 0 ,0
Exp/Cntr(USF)=0,0
Exp/Cntr=0.3,0.1

Type RM Length L Ch R = 1 ,50499   ,371.2,371.2,371.2
XS GIS Cut Line= 3
  2200308.620583 614054.05561121 2200418.2073302613976.418922605
2200684.72664051613539.664359132
#Sta/Elev= 30
       0 2444.24      43 2430.96    77.6 2418.78    97.9 2415.48   132.3 2406.12
   152.6 2404.31   184.7 2403.46  196.782400.131   210.8 2399.07  222.13 2400.13
   230.2 2401.13   237.9 2403.78   245.6  2404.8   259.9 2404.43   318.5 2406.13
   344.7 2404.43   372.4    2404   394.2 2406.55   422.2 2406.25     432 2405.38
   452.4 2405.86   456.7 2406.81   466.9 2412.32   475.5  2415.3   517.7 2421.01
   536.8 2425.42   555.1 2427.07   564.5  2431.2   606.5 2444.39     646 2459.91
#Mann= 8 ,-1,0
       0     .08       0      50      .1       0  196.78    .045       0
  222.13      .1       0   244.3     .05       0   354.3      .1       0
   374.3     .06       0   564.3      .1       0
Bank Sta=196.78,222.13
XS Rating Curve= 0 ,0
Exp/Cntr=0.3,0.1

Type RM Length L Ch R = 1 ,50128   ,277.8,277.8,277.8
XS GIS Cut Line= 3
2200501.59263515 614397.323409622200636.95511609 614344.15254228
2200966.28152405613769.471147595
#Sta/Elev= 30
       0 2433.37    32.9  2423.1    41.5 2419.08    54.6 2417.91   118.8  2404.7
   145.4 2395.36   155.6 2393.87   167.6 2392.82   208.6 2394.67   246.7 2393.62
   259.5 2391.17   273.3 2391.38   296.5 2395.44   347.1 2395.16   366.8 2396.43
   387.4 2395.05  400.68 2392.51  426.482392.548   443.9  2397.8   489.9 2393.84
   508.5 2398.05   557.3 2397.35   577.6 2397.04   642.3 2403.13   662.8 2403.16
   674.4 2407.97   702.1 2409.22   715.9    2413   747.2 2418.31   807.8 2432.47
#Mann= 6 ,-1,0
       0     .08       0   155.6      .1       0  400.68    .045       0
  426.48      .1       0   557.3     .06       0   747.2      .1       0
#XS Ineff= 2 , 0
           369.1    2398
Permanent Ineff=
       F       F
Bank Sta=400.68,426.48
XS Rating Curve= 0 ,0
Exp/Cntr=0.3,0.1

Type RM Length L Ch R = 1 ,49850   ,144.6,144.6,144.6
XS GIS Cut Line= 5
2200598.05760272614543.9888129132200776.11886258614342.041286478
2200923.77941955  614319.24075932200950.58614947614327.420331439
 2201300.1070173614326.355327227
#Sta/Elev= 30
       0 2432.13    37.5 2424.25   125.4 2410.46   142.4 2405.72   163.7 2393.99
   170.7 2392.26   214.9 2389.77   265.1 2394.75   284.1 2389.65   305.7 2387.42
   333.2  2386.7   358.3 2390.42   382.2 2386.52   389.2 2385.66  403.672386.487
     415 2388.88   431.6 2386.81   444.2 2389.47   456.3 2388.32   512.3 2389.26
   548.3  2388.2   576.3 2390.54   652.3 2389.95   676.3 2391.06   692.3 2397.98
   704.3 2408.92   724.3 2421.04   745.6 2422.58   756.3 2429.97   796.2  2444.6
#Mann= 6 ,-1,0
       0     .08       0      70      .1       0   382.2    .045       0
  403.67      .1       0  536.67     .08       0  726.67     .06       0
#XS Ineff= 2 , 0
          358.34    2395
Permanent Ineff=
       F       F
Bank Sta=382.2,403.67
XS Rating Curve= 0 ,0
Exp/Cntr(USF)=0,0
Exp/Cntr=0.3,0.1

Type RM Length L Ch R = 1 ,49705   ,219.4,219.4,219.4
XS GIS Cut Line= 3
2200651.99647546614601.2217236372200818.62097296614492.663338899
2201300.82217029614346.235750181
#Sta/Elev= 30
       0 2425.29    57.5 2417.02   105.2 2408.41   146.6 2399.01   176.9 2395.29
   182.3 2394.13   193.8 2389.12   204.7 2388.53   212.5 2386.87   225.6 2387.62
   242.3 2385.25   254.2 2387.39   263.2 2387.54  289.772384.027   309.2 2382.85
  318.652384.028   325.9 2385.65     344  2385.3   367.7 2386.47   418.1  2385.1
   447.1 2386.92   463.9 2385.59   481.9 2387.62   564.2 2389.41   589.3 2401.58
   618.5 2410.91   643.6 2422.96   664.5 2423.84   674.3 2431.82   702.8 2443.95
#Mann= 6 ,-1,0
       0     .08       0      40      .1       0  289.77    .045       0
  318.65      .1       0  428.87     .08       0  628.87     .06       0
Bank Sta=289.77,318.65
XS Rating Curve= 0 ,0
Exp/Cntr(USF)=0,0
Exp/Cntr=0.3,0.1

Type RM Length L Ch R = 1 ,49486   ,121.8,121.8,121.8
XS GIS Cut Line= 2
2200817.35841058614732.662849415 2201373.6824053614500.583578164
#Sta/Elev= 30
       0 2413.38    26.2 2408.03    50.7  2404.5    72.4 2399.59    94.1 2398.38
    98.4 2396.34   107.1 2387.23   111.4 2385.89   124.4 2385.85   132.6 2380.58
   148.6  2379.5  155.53  2380.6   163.4 2382.25   196.1 2380.71   202.4 2379.59
   211.1 2381.26   263.1 2382.65     300 2381.97   341.1 2384.97   427.8  2382.8
   471.1  2383.2   475.8 2384.52   488.5 2395.01   514.5 2409.78   536.1 2426.24
   553.5 2426.83   557.8 2429.48   562.2 2434.67   567.5 2438.72   602.8 2458.88
#Mann= 7 ,-1,0
       0      .1       0     130     .08       0   132.6    .045       0
  155.53      .1       0     240     .08       0     450     .06       0
     560      .1       0
Bank Sta=132.6,155.53
XS Rating Curve= 0 ,0
Exp/Cntr(USF)=0,0
Exp/Cntr=0.3,0.1

Type RM Length L Ch R = 1 ,49364   ,137.5,137.5,137.5
XS GIS Cut Line= 2
2200858.96010239614853.5431306932201381.92129322614571.170117124
#Sta/Elev= 30
       0 2406.33      15 2405.77    55.9 2399.02    78.7 2397.28   101.4 2393.89
     115 2384.18   128.7 2383.62   137.8 2378.27   142.9 2377.07   155.9 2379.59
  172.23 2378.37   192.3 2377.48   207.8 2378.43   222.6 2381.97   253.3 2380.74
   290.5 2383.07   322.9 2381.41   354.4 2383.62   393.8 2380.85   482.3 2381.25
   487.8 2384.22   519.6 2408.74   532.5 2413.39   544.3 2421.59     562 2423.34
   565.1  2424.9   573.8 2434.56   576.8 2436.52   588.6 2440.39   594.3 2443.58
#Mann= 6 ,-1,0
       0      .1       0     170     .08       0  172.23    .045       0
   207.8     .08       0     430     .06       0     580      .1       0
Bank Sta=172.23,207.8
XS Rating Curve= 0 ,0
Exp/Cntr=0.3,0.1

Type RM Length L Ch R = 1 ,49227   ,185.2,185.2,185.2
XS GIS Cut Line= 2
2200941.72624972614970.2942563422201423.65162638614624.951417304
#Sta/Elev= 30
       0 2400.89      14 2399.61    39.8 2393.59    68.5 2389.85    81.7 2382.87
    96.5 2381.61   106.4 2376.74   131.6 2377.77  148.11 2376.03   168.8 2375.11
  178.44 2376.03   197.5 2376.38   209.7 2380.03   239.2 2381.73     254 2379.92
     272 2381.04   297.2 2378.81   335.1 2381.24   367.2 2377.79   401.6 2379.58
   450.8  2379.8   470.5  2391.1   484.2 2402.98     500 2414.69     505 2417.27
     510 2417.87   541.5 2418.73     564  2436.2   583.7 2441.64   592.9 2449.61
#Mann= 7 ,-1,0
       0      .1       0  148.11    .045       0  178.44      .1       0
     240     .08       0     360     .06       0     480      .1       0
     510     .06       0
Bank Sta=148.11,178.44
XS Rating Curve= 0 ,0
Exp/Cntr(USF)=0,0
Exp/Cntr=0.3,0.1

Type RM Length L Ch R = 1 ,49041   ,361.2,361.2,361.2
XS GIS Cut Line= 3
2200952.02753233615143.0189452792201092.54154841615106.144443352
 2201518.9273068614727.139271971
#Sta/Elev= 30
       0 2404.95    33.2 2401.37   115.9 2388.59   128.4 2388.08   144.9  2378.1
   160.8 2376.77   176.8 2371.72   192.9 2374.38   241.1 2375.32     276 2373.63
   281.7 2371.76   289.3 2370.29  301.022371.822     310 2374.69   321.4 2374.25
   341.2 2376.35   383.7 2373.28     407 2375.88   491.4 2374.48   542.4 2377.39
   562.2 2385.28   583.6 2397.57     605 2412.61   610.3 2414.06   635.9 2414.49
   658.5 2430.22   674.6 2433.61     684 2441.44   694.6 2442.59   715.8 2452.99
#Mann= 7 ,-1,0
       0     .08       0      90      .1       0   281.7    .045       0
  301.02      .1       0  335.27     .08       0  495.27      .1       0
  595.27     .06       0
#XS Ineff= 2 , 0
                        349.3647            2380
Permanent Ineff=
       F       F
Bank Sta=281.7,301.02
XS Rating Curve= 0 ,0
Exp/Cntr=0.3,0.1

Type RM Length L Ch R = 1 ,48680   ,304,304,304
XS GIS Cut Line= 3
2201068.83253436615428.4316836222201240.23144393615441.918051962
2201733.67714796614940.811476318
#Sta/Elev= 30
       0 2401.51    35.5 2393.44   139.8 2377.29   163.8 2368.63   183.2 2367.43
     212 2369.21   291.6  2369.7   342.9 2368.53   371.4 2369.67   412.8 2367.87
   451.2 2368.14  457.762366.429     474 2364.82  483.01 2366.43   489.2 2369.37
   503.3 2368.32   543.5 2369.24   562.7  2367.9   588.4 2368.73   616.5 2366.78
   630.6 2369.67   650.1 2371.32   667.4 2379.11   684.9  2383.6   707.7 2396.85
   730.5 2398.06   773.6 2413.85   807.3 2429.51   856.9 2446.21   875.2 2455.27
#Mann= 9 ,-1,0
       0     .08       0      70      .1       0  281.93     .05       0
  421.93      .1       0  457.76    .045       0  483.01      .1       0
  561.93     .08       0  581.93     .06       0  721.93      .1       0
#XS Ineff= 2 , 0
        383.6376    2373
Permanent Ineff=
       F       F
Bank Sta=457.76,483.01
XS Rating Curve= 0 ,0
Exp/Cntr=0.3,0.1

Type RM Length L Ch R = 1 ,48376   ,397.2,397.2,397.2
XS GIS Cut Line= 2
2201213.34148089615792.0160818692201954.31557207615187.371125011
#Sta/Elev= 30
       0 2387.35    24.3  2379.4    81.1 2369.43   112.2 2361.18   168.9 2362.72
   246.3 2360.43   282.4 2363.68   344.4 2361.14   468.3 2363.37   499.3 2363.04
  506.882360.464   512.9 2359.58  534.612360.485   561.2 2364.09   656.1  2365.7
   677.8 2365.13   697.7 2361.55   711.9  2362.7   719.4 2366.22   731.8 2378.24
   737.5 2381.43   757.4 2388.07   778.1 2388.56   788.4 2393.87   803.9 2395.79
   886.5 2426.38   917.5 2435.36   927.8  2439.9   933.7  2440.4   956.4 2449.28
#Mann= 8 ,-1,0
       0     .08       0      30      .1       0     210     .05       0
     410      .1       0  506.88    .045       0  534.61      .1       0
     790     .06       0     830     .05       0
#XS Ineff= 2 , 0
        472.5322    2373
Permanent Ineff=
       F       F
Bank Sta=506.88,534.61
XS Rating Curve= 0 ,0
Exp/Cntr(USF)=0,0
Exp/Cntr=0.3,0.1

Type RM Length L Ch R = 1 ,47979   ,213.3,213.3,213.3
XS GIS Cut Line= 4
2201259.18443145615921.1910006712201441.04907831615813.176576146
2201991.25602681615810.5506755392202413.34156616615996.508295347
#Sta/Elev= 30
       0  2397.1    52.3 2384.76    89.5 2378.97   126.8 2376.74   149.6 2372.93
   177.9  2365.7   196.5 2358.15   418.7 2356.69   436.82352.642   446.7 2350.92
   459.8 2352.64   466.7 2354.38   522.7 2356.41   566.7 2355.97   606.7 2353.51
   626.7 2355.34   646.7 2359.18   666.7 2359.99   730.7  2357.5   761.7 2360.15
   810.8 2356.62   889.5  2354.8  1046.9 2355.65  1068.7 2357.06  1081.8 2354.92
  1090.6 2356.46  1105.6 2363.75  1115.5 2365.43  1164.9 2369.81    1223 2372.05
#Mann= 7 ,-1,0
       0      .1       0     200     .05       0   436.8    .045       0
   459.8     .05       0  691.52     .07       0  791.74     .05       0
 1121.74      .1       0
#XS Ineff= 2 , 0
                        528.9468            2360
Permanent Ineff=
       F       F
Bank Sta=436.8,459.8
XS Rating Curve= 0 ,0
Exp/Cntr=0.3,0.1

Type RM Length L Ch R = 1 ,47766   ,91.5,91.5,91.5
XS GIS Cut Line= 3
2201310.29349451616035.5330372562202282.26972996616007.762287671
2202371.89351271616086.025309227
#Sta/Elev= 30
       0 2393.05    37.9 2390.45    49.9 2388.17    85.9 2376.84   101.9 2373.47
   149.9 2364.28   165.9 2363.28     214 2353.72     266 2353.55     322 2350.45
     342 2350.72  354.962348.716     362 2347.66  379.532348.718     386 2351.33
   426.1 2352.13   462.1  2350.7   502.1 2352.25   526.1 2350.86   610.1 2352.61
   662.2 2350.47   846.2 2352.51   862.2 2350.88   950.3 2357.74   974.5 2366.04
  1025.8 2368.54  1038.6 2365.15  1048.4 2364.39  1065.7  2370.4  1091.4 2376.29
#Mann= 7 ,-1,0
       0      .1       0     220     .05       0  354.96    .045       0
  379.53     .05       0     610     .06       0     810     .05       0
     910      .1       0
#XS Ineff= 1 ,-1
606.50481091.358    2360
Permanent Ineff=
       F
Bank Sta=354.96,379.53
XS Rating Curve= 0 ,0
Exp/Cntr(USF)=0,0
Exp/Cntr=0.3,0.1

Type RM Length L Ch R = 1 ,47674   ,38.7,38.7,38.7
XS GIS Cut Line= 6
2201311.56167862616054.560861486 2201523.9168345616062.805148153
2201597.13062886616095.6251249342201673.98198296616119.594436574
2201770.06666036616238.2657932532202310.33397046616363.234166383
#Sta/Elev= 30
       0 2395.57    32.6 2390.32    41.6 2386.79    68.7 2381.72    93.7 2374.73
   152.7 2365.88   168.7 2361.41   196.8  2358.9   230.3 2353.17   312.7  2350.1
   329.5 2348.87   337.8 2346.51  359.65 2346.51   367.2 2348.95   427.6 2349.77
   556.8 2345.65   630.7 2348.21   675.9  2346.1   745.7 2347.19   790.9  2346.1
   823.7 2346.77     840 2345.44   848.3 2346.54   934.6 2345.51   959.2 2348.59
   987.9 2357.27  1024.9  2377.1  1041.3 2383.87  1061.8 2391.11  1080.5 2395.82
#Mann= 7 ,-1,0
       0      .1       0     120     .05       0   337.8    .045       0
  359.65     .05       0  585.94     .06       0  685.94     .05       0
  985.94      .1       0
#XS Ineff= 2 , 0
                          627.61            2360
Permanent Ineff=
       F       F
Bank Sta=337.8,359.65
XS Rating Curve= 0 ,0
Exp/Cntr=0.3,0.1

Type RM Length L Ch R = 1 ,47636   ,131.7,131.7,131.7
XS GIS Cut Line= 6
2201312.45566376616094.4888315362201524.81081964616102.733118203
  2201598.024614616135.553094984 2201674.8759681616159.522406624
 2201770.9606455616278.1937633032202306.37554925616397.500995693
#Sta/Elev= 30
       0 2399.04     7.7 2396.99    15.7 2392.71    31.7 2388.14    95.8 2373.41
   135.8 2367.34   155.8 2362.07     168 2361.13     195 2356.12   255.7 2351.46
   320.1 2349.97  334.83 2346.09   345.3 2345.09  351.64 2346.06     362 2348.84
   457.7 2349.17   547.7 2346.88   568.2 2345.32   633.7 2347.46   715.7 2344.38
   748.5 2346.42   831.1 2345.04   850.9 2346.16   908.3 2344.69   945.2 2345.68
   965.7 2352.77   982.1 2362.29   994.4 2365.32  1035.5 2384.02  1074.5 2398.43
#Mann= 7 ,-1,0
       0      .1       0     120     .05       0  334.83    .045       0
  351.64     .05       0  503.25     .06       0  685.94     .05       0
  885.94      .1       0
Bank Sta=334.83,351.64
XS Rating Curve= 0 ,0
Exp/Cntr=0.3,0.1

Type RM Length L Ch R = 1 ,47504   ,300.2,300.2,300.2
XS GIS Cut Line= 3
2201375.93344807616335.9620554862201702.87090909616271.584408722
2202301.20433195616401.602009049
#Sta/Elev= 30
       0 2380.02    28.8  2373.3    57.1 2368.42    76.5  2363.1    85.9 2362.93
   102.2 2360.37     147 2360.07   228.5  2348.4   281.5 2349.77  289.31 2344.61
   293.8 2343.41   310.1 2344.57   319.3 2349.24   371.4  2348.9   445.1 2345.19
   510.6 2347.66   596.5 2344.24   625.2 2346.28   695.5 2345.59     703 2344.56
   725.1 2346.07   780.7 2344.61   817.6 2345.01   825.8 2346.58   842.1 2353.85
   858.5 2362.71   874.9 2367.66   887.2 2372.91   895.3 2377.82   945.5 2397.27
#Mann= 7 ,-1,0
       0      .1       0     160     .05       0  289.31    .045       0
   310.1     .05       0  353.22     .06       0  563.22     .05       0
  763.22      .1       0
#XS Ineff= 2 , 0
                        494.4732            2360
Permanent Ineff=
       F       F
Bank Sta=289.31,310.1
XS Rating Curve= 0 ,0
Exp/Cntr(USF)=0,0
Exp/Cntr=0.3,0.1

Type RM Length L Ch R = 1 ,47204   ,361.1,361.1,361.1
XS GIS Cut Line= 3
2201422.19902853616588.9911097042202165.64121553616515.568201067
2202301.29753868 616563.92410669
#Sta/Elev= 30
       0 2378.43    12.6 2376.75    82.1 2357.65   102.5 2359.53   134.6 2356.91
   158.9 2356.52   188.2 2352.77     215  2351.2   231.1 2343.81  236.792339.631
   251.2  2338.1  261.46 2339.63   267.3 2342.58   271.3 2342.83   327.6  2341.5
   391.9 2342.79     420 2341.53   480.3 2343.83   586.9 2342.56     617 2341.05
   677.3 2343.09   689.3 2341.41     715 2342.62   736.9 2346.16   756.6 2351.59
   792.2  2367.5   809.2 2377.67   847.4 2393.82   855.9    2397   891.1 2405.82
#Mann= 6 ,-1,0
       0     .08       0  236.79    .045       0  261.46     .08       0
     400     .06       0     420     .05       0  807.06      .1       0
#XS Ineff= 2 , 0
                        388.6266            2360
Permanent Ineff=
       F       F
Bank Sta=236.79,261.46
XS Rating Curve= 0 ,0
Exp/Cntr=0.3,0.1

Type RM Length L Ch R = 1 ,46843   ,372.6,372.6,372.6
XS GIS Cut Line= 2
2201464.35966037616894.2602408532202207.71810884616928.545116883
#Sta/Elev= 30
       0  2371.8    31.8 2368.09    55.9 2363.52    79.9 2360.56   119.9 2357.44
     164 2349.72     176 2346.75     188 2339.48     196 2338.92   203.3 2334.21
     208 2332.94   231.8 2334.21   248.1 2336.66   276.1 2337.26   300.1 2335.71
   376.2 2334.43   408.1 2337.03   460.3 2337.17   516.4 2336.57   524.4 2335.37
   532.4 2332.46   544.4 2334.14   588.3 2335.92   612.5 2338.85   620.5 2342.65
   636.5 2355.44   653.3 2366.79   680.5 2376.15   724.6 2384.42   744.1 2394.36
#Mann= 6 ,-1,0
       0     .08       0   203.3    .045       0   231.8     .08       0
     260     .06       0     360     .05       0     560      .1       0
#XS Ineff= 2 , 0
                        281.6483            2340
Permanent Ineff=
       F       F
Bank Sta=203.3,231.8
XS Rating Curve= 0 ,0
Exp/Cntr(USF)=0,0
Exp/Cntr=0.3,0.1
